--- LBngmnCrk.prj (project) ---

Proj Title=LBngmnCrk
Current Plan=p01
Default Exp/Contr=0,0
English Units
Geom File=g01
Flow File=f01
Plan File=p01
BEGIN DESCRIPTION:
END DESCRIPTION:
DSS Export Rating Curves= 0
DSS Export Rating Curve Sorted= 0
DSS Export Volume Flow Curves= 0
DXF OffsetX= 0
DXF OffsetY= 0
DXF ScaleX= 0
DXF ScaleY= 0

--- LBngmnCrk.p01 (plan) ---

Plan Title=Floodplain
Program Version=4.00
Geom File=g01
Flow File=f01
K Sum by GR=0
Std Step Tol=0.01
Critical Tol=0.01
Num of Std Step Trials=20
Max Error Tol=0.3
Flow Tol Ratio=0.001
Split Flow NTrial=30
Split Flow Tol=0.02
Split Flow Ratio=0.02
Log Output Level=0
Friction Slope Method=1
Unsteady Friction Slope Method=2
Unsteady Bridges Friction Slope Method=1
Global Log Level=0
CheckData=False
Run HTab=0
Run UNet=0
Run PostProcess=0
UNET Theta=0
UNET Theta Warmup=0
UNET ZTol=0
UNET ZSATol=0
UNET MxIter=0
UNET MaxInSteps=0
UNET DtIC=0
UNET DtMin=0
UNET MaxCRTS=0
UNET WFStab=0
UNET SFStab=0
UNET WFX=0
UNET SFX=0
UNET DSS MLevel=0
UNET DZMax Abort=0
UNET Convert EG Bridges=0
UNET Use Existing IB Tables=0
UNET Froude Limit=0
UNET Froude Power=0
Write IC File=0
Echo Input=False
Echo Output=False
Write Detailed=0

--- LBngmnCrk.f01 (steady flow) ---

Flow Title=NFF Regression Equation
Program Version=4.00
Number of Profiles= 1
Profile Names=P100yr
River Rch & RM=LBngmnCrk,Main            ,32609.5
  747.42
River Rch & RM=LBngmnCrk,Main            ,31810.1
  768.17
River Rch & RM=LBngmnCrk,Main            ,31334.6
965.1096
River Rch & RM=LBngmnCrk,Main            ,29502.3
1010.117
River Rch & RM=LBngmnCrk,Main            ,27423.2
 1121.86
River Rch & RM=LBngmnCrk,Main            ,27098.4
  1299.6
River Rch & RM=LBngmnCrk,Main            ,25473.1
1322.422
River Rch & RM=LBngmnCrk,Main            ,25054.6
1469.992
River Rch & RM=LBngmnCrk,Main            ,23931.1
 1552.82
River Rch & RM=LBngmnCrk,Main            ,23514.1
1801.185
River Rch & RM=LBngmnCrk,Main            ,17114.1
1944.272
River Rch & RM=LBngmnCrk,Main            ,15114.1
2222.824
River Rch & RM=LBngmnCrk,Main            ,7574.6
2457.074
River Rch & RM=LBngmnCrk,Main            ,1914.1
2729.139
River Rch & RM=LBngmnCrk,Main            ,1451.2
6086.096
River Rch & RM=LBngmnCrk,Main            ,265.6
6986.264
Boundary for River Rch & Prof#=LBngmnCrk,Main            , 1
Up Type= 0
Dn Type= 3
Dn Slope=0.00525
DSS Import GetInterval= 0
DSS Import GetPeak= 0
DSS Import FillOption= 0

--- LBngmnCrk.g01 (geometry) ---

Geom Title=USGS 3m DEM
Program Version=4.00

River Reach=LBngmnCrk       ,Main
Reach XY= 30
     1726814.178      359263.616     1727630.239      358730.048
     1728662.621      357482.259     1730529.951      354427.901
     1731216.035      353795.292     1731339.019      352481.973
     1731510.562      351958.307     1731814.774      351848.302
     1731643.842      351567.609     1732026.203       350624.91
     1733035.537      350257.087     1733341.304      349382.655
     1734415.504       349055.38     1735411.193      347423.924
     1737960.468      345621.719     1738636.672      345424.155
     1739086.667      345780.162     1739331.507      345448.339
     1739832.229       345482.35     1740095.918      345049.979
     1741659.468      344819.793     1741995.901      344528.821
     1742109.564      343896.187     1743563.508      342593.576
     1743274.453      342023.445       1744024.5      341882.891
     1743989.496      341362.408     1744358.727      341281.107
     1745109.668      341862.933     1745358.762      341364.027

Type RM Length L Ch R = 1 ,32609.5 ,410.581,400,394.436
XS GIS Cut Line= 3
     1726954.795      359707.727     1726822.957      359258.828
     1726606.165      358861.378
#Sta/Elev= 30
       0 1191.69     117 1154.72   146.2 1140.78   185.2 1126.73   243.7 1118.25
   272.9 1110.52   302.2 1106.26   321.7 1101.51   341.1 1089.94   360.6 1084.92
   380.1 1082.74   438.6 1082.59   460.4 1079.44   467.9 1079.43   475.4 1080.61
   525.7 1087.51   573.8 1090.47   602.7 1100.82   631.6 1107.15   650.9 1116.59
   670.1 1120.05   689.4 1129.05   708.7 1133.03   737.6 1145.38   795.4 1158.81
   814.6 1167.78   872.4 1184.79   882.1 1184.69   891.7 1188.62   920.6 1194.71
#Mann= 3 , 0 , 0
       0      .1       0   460.4    .045       0   475.4      .1       0
Bank Sta=460.4,475.4
XS Rating Curve= 0 ,0
Exp/Cntr=0.3,0.1

Type RM Length L Ch R = 1 ,32209.5 ,397.224,399.465,401.173
XS GIS Cut Line= 3
      1727457.82       359405.13     1727147.026      359073.298
     1726839.367      358736.967
#Sta/Elev= 30
       0 1194.79    48.4 1182.68    67.7 1180.11   116.1 1163.79   135.4 1154.73
   145.1 1146.28   154.8  1140.7   222.5 1135.12   241.8 1130.14   290.2 1108.03
   309.5 1095.14   338.6  1092.1   367.6 1083.83     445 1076.11   447.1 1076.11
   462.1 1076.11   493.4  1076.4   503.1 1079.12   561.3 1102.87   580.7 1114.28
   609.8 1127.45   638.9 1145.48   658.3 1150.01   687.4 1166.41   706.8 1170.61
   745.6 1186.18     765 1190.84   784.4 1198.85     862 1217.19   910.5 1220.47
#Mann= 3 , 0 , 0
       0      .1       0   447.1    .045       0   462.1      .1       0
Bank Sta=447.1,462.1
XS Rating Curve= 0 ,0
Exp/Cntr=0.3,0.1

Type RM Length L Ch R = 1 ,31810.1 ,479.241,475.499,472.024
XS GIS Cut Line= 3
     1727738.412      359190.357     1727460.382      358828.615
     1727172.045      358477.275
#Sta/Elev= 30
       0 1190.94    87.4 1173.85   126.2 1156.15   213.6 1133.57   262.1 1115.72
   271.8 1108.66   291.2 1103.28   320.3 1084.94     330 1081.03     398  1075.4
   434.5 1069.66   436.8 1069.55   449.5  1069.9   456.2 1070.68   465.9 1076.46
   475.6 1085.33   504.6 1098.37   523.9 1109.91   591.6 1130.71   620.6 1144.79
     640 1148.66     669 1162.48   688.3 1166.45   717.3 1182.22   765.7  1197.5
   794.7 1203.13   823.7 1214.63   843.1 1218.05   872.1 1227.03   910.8 1232.16
#Mann= 3 , 0 , 0
       0      .1       0   434.5    .045       0   449.5      .1       0
Bank Sta=434.5,449.5
XS Rating Curve= 0 ,0
Exp/Cntr=0.3,0.1

Type RM Length L Ch R = 1 ,31334.6 ,329.184,323.708,319.672
XS GIS Cut Line= 3
     1728112.572      358845.904     1727892.565      358587.787
      1727505.13      358291.157
#Sta/Elev= 30
       0 1083.28    29.1 1082.47    48.5 1079.39   106.6 1079.53   116.3 1080.11
   135.7  1084.6   145.4 1085.52   213.2 1081.64   242.3 1076.38   271.3 1075.75
   290.7 1072.86   339.2 1069.55     472 1069.44     487 1068.25   495.3 1066.48
   505.1 1066.27   514.8 1067.95   524.6 1072.78   534.3 1080.21   544.1 1083.35
   612.4 1116.42   641.7 1127.24   690.5 1140.06   719.8 1150.35   729.5  1151.5
     749 1157.04   778.3 1160.86   797.8 1166.38   817.3 1168.86   827.1 1171.79
#Mann= 3 , 0 , 0
       0      .1       0     472    .045       0     487      .1       0
Bank Sta=472,487
XS Rating Curve= 0 ,0
Exp/Cntr=0.3,0.1

Type RM Length L Ch R = 1 ,31010.9 ,383.967,394.195,402.984
XS GIS Cut Line= 3
     1728277.455      358440.761     1727868.006      358197.673
     1727503.055       357932.25
#Sta/Elev= 30
       0 1196.54    19.4 1188.55    38.9 1182.89    48.6  1177.8      68 1173.04
    87.5 1164.95   106.9 1159.29     136 1145.09   145.8 1144.87   194.4 1125.35
   213.8 1120.53   233.2 1111.19   281.8 1093.58   330.4 1073.04   388.7 1063.34
   460.9 1062.98   475.9 1063.72   495.8  1075.5     535 1092.08   564.5 1108.34
   574.3 1110.31   623.3 1135.74   642.9 1140.76     692 1160.62   721.4 1169.73
   770.5 1190.94   819.5 1205.87     898 1223.27   917.6 1225.07   927.4 1227.76
#Mann= 3 , 0 , 0
       0      .1       0   460.9    .045       0   475.9      .1       0
Bank Sta=460.9,475.9
XS Rating Curve= 0 ,0
Exp/Cntr=0.3,0.1

Type RM Length L Ch R = 1 ,30616.7 ,405.913,401.401,396.89
XS GIS Cut Line= 3
     1728425.415      358323.496     1728174.122      357944.185
     1727922.828      357564.874
#Sta/Elev= 30
       0 1203.73      29 1192.57    48.4 1189.94    77.4 1178.77    96.8 1174.83
   116.2 1164.55   154.9 1150.82   164.6 1144.59   280.7 1098.11   300.1 1085.21
   309.8 1080.89   338.8 1074.63   358.2 1063.25   367.9 1059.74   416.3 1056.43
   435.3 1056.43   450.3 1057.56   464.7 1064.18   493.7 1087.03   513.1 1094.28
   542.1 1111.69   590.5 1130.15   619.6  1138.1   638.9 1146.88   658.3 1150.78
   687.3 1166.53     697 1169.32   716.4 1179.62   764.8  1199.9     910 1243.25
#Mann= 3 , 0 , 0
       0      .1       0   435.3    .045       0   450.3      .1       0
Bank Sta=435.3,450.3
XS Rating Curve= 0 ,0
Exp/Cntr=0.3,0.1

Type RM Length L Ch R = 1 ,30215.3 ,311.248,305.751,300.253
XS GIS Cut Line= 3
     1728798.956       358006.52     1728477.223      357684.786
     1728155.489      357363.053
#Sta/Elev= 30
       0  1194.5     9.7 1194.41    38.7 1185.62    58.1 1182.33   145.2 1155.69
   183.9 1137.45   222.7 1123.58   261.4 1103.59   280.7  1097.5   309.8 1083.97
   329.1 1078.99   358.2 1065.87   377.6 1061.07   445.3 1053.03   447.5 1053.04
   462.5 1054.12     484 1062.79   493.7  1074.2   503.4 1080.11   542.1  1089.9
   619.6    1115   648.6 1133.91     668 1141.64   677.7 1148.64   735.7 1166.66
   764.8 1182.33   793.8 1193.45   842.2 1215.73   861.6 1221.54     910  1230.2
#Mann= 3 , 0 , 0
       0      .1       0   447.5    .045       0   462.5      .1       0
Bank Sta=447.5,462.5
XS Rating Curve= 0 ,0
Exp/Cntr=0.3,0.1

Type RM Length L Ch R = 1 ,29909.5 ,407.735,407.185,406.634
XS GIS Cut Line= 3
     1729249.381      357591.481     1728812.227      357537.511
     1728274.292      357214.263
#Sta/Elev= 30
       0 1158.75    19.6  1157.1    58.7 1167.03    88.1 1171.26   166.4 1159.45
   225.1 1142.06   244.7 1132.27   274.1 1121.21   283.9 1119.94   332.8 1098.94
   342.6 1096.94   362.2 1086.83     372 1085.23   411.1 1070.28   518.9 1054.16
   577.8 1054.95   597.2 1049.91   607.2 1049.87   612.2 1049.87   646.4 1054.16
     666 1071.07   695.4 1086.52   783.7 1118.03   822.9 1129.32   862.1 1145.99
   901.4 1158.23     970 1189.53   989.6 1202.93  1028.8 1221.99  1068.1 1231.42
#Mann= 3 , 0 , 0
       0      .1       0   597.2    .045       0   612.2      .1       0
Bank Sta=597.2,612.2
XS Rating Curve= 0 ,0
Exp/Cntr=0.3,0.1

Type RM Length L Ch R = 1 ,29502.3 ,442.624,443.493,444.118
XS GIS Cut Line= 3
      1729228.78      357240.647      1728876.99       357111.15
      1728396.66      356835.904
#Sta/Elev= 30
       0 1182.82    48.1 1174.19    86.5 1163.83   153.8 1140.41     173 1131.02
   182.6 1129.32   230.7 1109.88   307.6 1086.09   365.3  1052.5   374.9 1049.87
   423.4 1049.87   457.3 1046.59   472.3 1046.56   481.7  1046.2   510.8 1052.84
   530.3 1053.15     540 1056.91   549.7  1063.6   569.1  1083.9   578.8  1091.1
   598.3 1097.01   617.7 1107.58   666.2 1125.35   685.7 1136.59   705.1 1141.51
   724.5 1151.75   734.2 1153.79   763.4 1166.52   860.5 1187.67   928.5 1186.46
#Mann= 3 , 0 , 0
       0      .1       0   457.3    .045       0   472.3      .1       0
Bank Sta=457.3,472.3
XS Rating Curve= 0 ,0
Exp/Cntr=0.3,0.1

Type RM Length L Ch R = 1 ,29058.8 ,416.43,414.582,412.745
XS GIS Cut Line= 3
     1729456.437      356997.113     1728992.317      356723.254
     1728534.255       356516.42
#Sta/Elev= 30
       0 1175.27    58.8 1175.23    88.2 1171.54   137.2 1170.44   186.2    1164
     245 1138.88   264.5 1134.23   284.1 1124.03   333.1 1108.31   362.5 1093.72
   372.3 1085.54   411.5 1064.73   431.1 1049.49   446.2 1041.84   460.5 1040.02
   461.2 1040.02   489.9 1043.09   529.1 1043.31   548.6 1046.33   674.2 1046.84
   703.2 1055.33   732.2 1080.94   761.2    1092   809.5 1087.02   838.5 1091.91
   857.8 1090.92   915.8 1077.85   944.8 1074.04   973.8  1073.3  1041.5 1064.73
#Mann= 3 , 0 , 0
       0      .1       0   446.2    .045       0   461.2      .1       0
Bank Sta=446.2,461.2
XS Rating Curve= 0 ,0
Exp/Cntr=0.3,0.1

Type RM Length L Ch R = 1 ,28644.3 ,434.79,432.556,431.742
XS GIS Cut Line= 3
     1729886.224      356663.201     1729454.467      356528.277
     1728947.151      356280.016
#Sta/Elev= 30
       0 1190.32     9.8 1190.89    29.5 1188.08     118 1183.06   167.2 1173.85
     177 1173.87   196.7 1167.53   206.5 1166.46   226.2 1158.84   275.3 1146.23
   363.8 1112.19   373.7 1109.96   422.8    1091   462.1 1078.21   481.6 1068.23
   491.3 1065.04   510.8 1052.43   520.5  1043.9     540 1037.38   549.7 1036.74
   551.4 1036.91   566.4 1039.15   588.7 1043.31   773.7 1043.31   802.9 1047.33
   841.9 1062.53   890.6  1089.3   939.2 1096.18   958.7 1104.11  1017.2 1120.93
#Mann= 3 , 0 , 0
       0      .1       0   551.4    .045       0   566.4      .1       0
Bank Sta=551.4,566.4
XS Rating Curve= 0 ,0
Exp/Cntr=0.3,0.1

Type RM Length L Ch R = 1 ,28211.7 ,393.689,395.523,395.118
XS GIS Cut Line= 3
     1729866.673      356248.105     1729407.059      356067.606
     1729006.216      355867.186
#Sta/Elev= 30
       0 1170.08    58.1 1155.16    87.1 1140.44   135.5 1125.83   203.3 1094.81
   261.4 1072.77   290.5 1057.11   329.2 1041.17   348.6 1037.29     426 1033.46
   435.7 1030.62   464.7 1030.15   479.4 1027.53   484.1  1026.9   494.4 1027.86
   503.5 1032.52   513.3 1041.37   542.5 1057.85   552.2 1061.62   581.5 1080.86
   610.7 1095.54   659.4  1113.5   678.9 1123.07   698.4 1127.85   756.8 1159.54
   786.1 1178.07   795.8 1180.68   815.3 1190.02   844.5 1198.21   941.9  1213.8
#Mann= 3 , 0 , 0
       0      .1       0   479.4    .045       0   494.4      .1       0
Bank Sta=479.4,494.4
XS Rating Curve= 0 ,0
Exp/Cntr=0.3,0.1

Type RM Length L Ch R = 1 ,27816.2 ,382.925,392.952,405.124
XS GIS Cut Line= 3
     1730054.498      355954.585     1729643.903      355754.416
     1729227.783      355569.706
#Sta/Elev= 30
       0  1156.3    38.9 1139.74    77.8 1129.32   145.8 1103.77   174.9 1091.01
   204.1 1073.47   213.8 1070.35   233.3 1059.23   301.3 1033.72   340.2 1032.86
   398.5 1024.56   447.1 1020.34   449.3 1020.51   464.3 1022.63   495.5 1027.69
   524.6 1038.99   582.7 1066.92   602.1 1073.39   640.8  1080.6   669.9 1084.71
   679.6 1084.36     699 1089.91     728 1095.04   776.4 1099.12   795.8 1105.75
   805.5 1107.27   853.9 1108.76     883 1112.66   902.4 1118.04   912.1 1118.18
#Mann= 3 , 0 , 0
       0      .1       0   449.3    .045       0   464.3      .1       0
Bank Sta=449.3,464.3
XS Rating Curve= 0 ,0
Exp/Cntr=0.3,0.1

Type RM Length L Ch R = 1 ,27423.2 ,328.974,324.855,319.4
XS GIS Cut Line= 3
     1730194.719      355825.808     1729906.558      355474.234
     1729638.613      355103.546
#Sta/Elev= 30
       0 1178.19    19.3 1168.12    48.4 1159.26    67.7 1149.34    96.7 1139.71
   116.1 1129.34   135.4 1123.58   164.4 1108.31   183.8 1101.09   212.8 1080.12
   232.1 1070.96   270.8 1041.65   290.2 1033.05   299.8 1030.38   328.8 1030.14
   348.2 1027.15   449.7 1021.83   464.3 1020.34   464.7 1020.34   483.8 1021.02
   493.5 1024.66   522.7 1042.66   542.2 1047.12     620 1084.21   668.7 1101.89
   717.3 1125.13   746.5 1133.62   775.7    1147     873 1182.54     912 1199.82
#Mann= 3 , 0 , 0
       0      .1       0   449.7    .045       0   464.7      .1       0
Bank Sta=449.7,464.7
XS Rating Curve= 0 ,0
Exp/Cntr=0.3,0.1

Type RM Length L Ch R = 1 ,27098.4 ,442.901,432.496,422.09
XS GIS Cut Line= 3
     1730544.655      355659.364     1730247.822      355340.943
     1729837.652      354984.742
#Sta/Elev= 30
       0 1084.25    96.7 1089.23   116.1 1087.86   145.1 1091.12   164.5 1089.19
   183.8 1093.44   212.8  1089.5   241.8 1090.65   270.9 1083.38   290.2 1084.07
   309.6 1081.02   348.3 1065.52   357.9 1058.25   406.3 1032.64   503.2 1023.62
   532.3 1023.62   619.6 1017.06   621.3 1017.06   636.3 1017.61   706.9 1038.24
     736 1050.23   765.1 1057.72   774.8 1062.99   794.3  1068.4   842.8 1089.44
   852.5 1095.46   871.9  1101.8     901 1118.68   920.4 1124.46   978.6 1153.81
#Mann= 3 , 0 , 0
       0      .1       0   621.3    .045       0   636.3      .1       0
Bank Sta=621.3,636.3
XS Rating Curve= 0 ,0
Exp/Cntr=0.3,0.1

Type RM Length L Ch R = 1 ,26665.9 ,377.691,399.394,422.649
XS GIS Cut Line= 3
     1730796.315      354965.537     1730356.049      354850.685
     1729915.783      354735.833
#Sta/Elev= 30
       0  1176.1    48.4 1157.14    96.8 1142.88   125.9 1128.18   145.2 1115.95
   164.6 1107.38   193.6 1089.83     213  1075.1   222.7 1072.02     242 1057.82
   251.7  1055.7   271.1 1043.86   290.4 1040.55   300.1 1033.79   319.5 1025.34
   396.9 1020.34   445.3 1020.33   474.4 1017.06   489.8 1017.06   504.8 1017.06
   542.1 1020.91     668 1046.88   735.7 1058.19   784.1 1074.03   832.6 1095.79
   851.9 1101.67   871.3 1113.91     881 1115.74   900.3 1127.04     910 1129.87
#Mann= 3 , 0 , 0
       0      .1       0   489.8    .045       0   504.8      .1       0
Bank Sta=489.8,504.8
XS Rating Curve= 0 ,0
Exp/Cntr=0.3,0.1

Type RM Length L Ch R = 1 ,26266.5 ,392.887,379.249,364.06
XS GIS Cut Line= 3
      1730848.39      354862.795     1730512.659      354510.324
     1730325.418      354101.797
#Sta/Elev= 30
       0 1157.39    58.4 1140.63   116.8 1115.11   126.6 1113.95   155.8 1100.28
   175.2 1093.91   204.4 1078.45   223.9  1071.8   243.4 1059.08   282.3 1042.38
   311.5 1037.68   360.2 1021.79   399.2 1017.06   438.1 1017.06   486.8 1012.17
   504.4 1013.32   519.4 1014.85   545.4 1018.08   584.5 1034.53     604 1047.08
   623.5 1052.66   672.4 1078.51   701.7 1088.57     731 1106.95   760.3 1118.26
   818.9 1147.49   838.5 1153.85     858 1165.54   906.9 1181.79   936.2 1188.24
#Mann= 3 , 0 , 0
       0      .1       0   504.4    .045       0   519.4      .1       0
Bank Sta=504.4,519.4
XS Rating Curve= 0 ,0
Exp/Cntr=0.3,0.1

Type RM Length L Ch R = 1 ,25887.2 ,412.769,414.098,415.426
XS GIS Cut Line= 3
     1731196.769      354523.146     1730816.222      354273.822
     1730443.612      354012.198
#Sta/Elev= 30
       0  1087.9      29 1080.73    58.1 1080.51    87.1 1076.44   106.5 1077.69
   135.5 1072.86   193.6 1054.75   222.6 1039.86   232.3 1036.74   251.7 1036.01
   290.4 1023.87   309.8 1023.62   358.2 1017.13   464.6 1016.85   483.2 1012.45
   498.2 1010.62   503.4  1010.5   522.8  1011.1   532.4 1013.45   561.5 1028.57
   580.9 1041.08   609.9  1050.6   648.7 1069.39   668.1  1076.4   706.8 1095.86
   755.2  1111.6   774.6 1122.87   803.7 1131.63   842.4 1149.66   910.2 1173.58
#Mann= 3 , 0 , 0
       0      .1       0   483.2    .045       0   498.2      .1       0
Bank Sta=483.2,498.2
XS Rating Curve= 0 ,0
Exp/Cntr=0.3,0.1

Type RM Length L Ch R = 1 ,25473.1 ,425.536,418.513,411.491
XS GIS Cut Line= 3
     1731402.095      354231.716       1731046.8       353947.48
     1730691.505      353663.244
#Sta/Elev= 30
       0 1112.32    77.4 1094.75   116.2 1080.23   135.5 1075.12   183.9 1052.33
   203.3 1047.56     213 1042.92   232.3 1028.28   251.7 1021.63   309.8 1017.06
   358.2 1016.92   367.9 1014.28   416.3 1013.56   449.1 1009.33     455 1007.66
   464.1 1007.75   474.4 1012.11   493.7 1030.98   503.4 1037.24   571.2 1057.24
   580.9 1064.39   619.6 1085.25   638.9 1091.54     668 1107.65   706.7    1119
   745.4 1134.55   764.8 1138.87   822.9 1161.25   832.6 1162.56     910  1189.6
#Mann= 3 , 0 , 0
       0      .1       0   449.1    .045       0   464.1      .1       0
Bank Sta=449.1,464.1
XS Rating Curve= 0 ,0
Exp/Cntr=0.3,0.1

Type RM Length L Ch R = 1 ,25054.6 ,405.619,401.711,397.804
XS GIS Cut Line= 3
     1731678.357      353768.449     1731251.921      353609.774
     1730825.485        353451.1
#Sta/Elev= 30
       0  1092.4    67.8 1074.39    77.4 1074.23   135.5 1054.23   154.9 1050.72
   174.3 1040.75   183.9 1038.46   203.3 1027.22     213 1024.21   300.1 1013.79
   338.8 1013.78   358.2 1010.97   406.6 1010.02     439 1003.38   445.3 1002.46
     454 1004.32   474.4 1009.73   503.4 1011.12   513.1  1014.3   580.9 1054.63
     668 1089.39   687.3 1099.18     697  1100.9   716.4 1109.58   755.1 1122.32
   784.1 1135.99   813.2 1146.72   822.9 1148.23   842.2    1156     910 1170.97
#Mann= 3 , 0 , 0
       0      .1       0     439    .045       0     454      .1       0
Bank Sta=439,454
XS Rating Curve= 0 ,0
Exp/Cntr=0.3,0.1

Type RM Length L Ch R = 1 ,24652.9 ,312.672,310.707,308.742
XS GIS Cut Line= 3
     1731840.794      353278.855     1731388.883      353234.345
     1730937.878      353144.382
#Sta/Elev= 30
       0 1150.43      58 1141.45   115.9 1123.51   144.9 1109.99   183.6 1094.97
   202.9 1084.52   212.6 1081.66   231.9 1071.14   241.5 1068.07   260.9 1056.38
   280.2 1049.31   309.2  1031.2   318.8  1020.7   328.5  1014.9   376.8  1013.7
   405.8  1010.5   454.1  1010.5   473.7 1007.32   532.4 1007.21   559.9  998.96
   561.7  998.34   574.9 1000.02   581.3 1001.54   591.1 1008.64   600.9  1019.4
   630.2 1041.46   659.6 1056.77   737.9 1084.06   816.1 1118.64     914 1150.86
#Mann= 3 , 0 , 0
       0      .1       0   559.9    .045       0   574.9      .1       0
Bank Sta=559.9,574.9
XS Rating Curve= 0 ,0
Exp/Cntr=0.3,0.1

Type RM Length L Ch R = 1 ,24342.2 ,411.523,411.16,410.796
XS GIS Cut Line= 3
     1731630.711      352948.786     1731399.663      352914.482
     1730955.726      352866.052
#Sta/Elev= 30
       0 1030.25    29.2 1018.18    58.4 1017.04    77.9 1013.78    97.3 1013.69
   116.8  1010.5   136.3  1010.2     146 1007.91   184.9 1003.93   223.8  1003.9
   243.3 1000.74   291.8    1003   311.2 1002.27   329.8  995.83   340.4  994.09
   344.8  995.02   379.2 1007.02   398.6 1020.53     418  1037.5   427.7 1043.43
   447.2 1051.44   466.6 1057.12   515.1 1076.59   553.9 1088.72   573.4 1097.29
   602.5 1107.12   641.3 1118.81     651 1119.37   670.4 1125.34   680.2 1125.78
#Mann= 3 , 0 , 0
       0      .1       0   329.8    .045       0   344.8      .1       0
#XS Ineff= 2 , 0
          291.98 1003.16
Permanent Ineff=
       F       F
Bank Sta=329.8,344.8
XS Rating Curve= 0 ,0
Exp/Cntr=0.3,0.1

Type RM Length L Ch R = 1 ,23931.1 ,404.545,416.912,417.626
XS GIS Cut Line= 3
     1731823.738      352539.913     1731305.628      352491.341
     1730933.237       352545.31
#Sta/Elev= 30
       0 1106.42    19.6 1101.71    39.3 1094.03    49.1  1091.7    68.7 1083.18
   127.6  1065.9   137.5 1064.57   176.7 1051.75   206.2 1037.87   255.3 1005.63
   314.2 1000.72   382.9 1000.65   412.4  997.37   461.5  997.18   480.7  994.02
   490.9  992.21   495.7   993.2   520.4 1000.63   636.2 1000.65   665.1 1003.75
   674.8 1007.18   684.4 1007.22     694 1011.31   703.7 1020.08   713.3 1026.66
   742.3 1035.87   761.6 1039.63   838.8 1043.28   858.1 1040.96   896.7 1042.52
#Mann= 3 , 0 , 0
       0      .1       0   480.7    .045       0   495.7      .1       0
Bank Sta=480.7,495.7
XS Rating Curve= 0 ,0
Exp/Cntr=0.3,0.1

Type RM Length L Ch R = 1 ,23514.1 ,1294.484,1278.392,1276.974
XS GIS Cut Line= 3
      1731877.52      352388.719     1731476.229      352102.237
     1731026.789      352046.631
#Sta/Elev= 30
       0 1128.51    19.3 1123.83    67.7 1105.21    96.7 1097.39   164.4 1072.12
   183.7  1061.6     203 1055.33     261 1024.51   280.4 1017.56   309.4 1001.44
     319  998.43     377  996.86   396.4  994.09   444.7  994.05   473.7  990.81
   485.6  990.82   500.6  991.15   512.3  993.51   541.2   994.1   550.9  997.24
   579.8  997.37   608.7  1000.6   647.2 1000.65     705 1007.22   791.8 1010.98
     811 1014.03   839.9 1021.02   888.1 1042.55   907.4 1046.73   945.9 1063.28
#Mann= 3 , 0 , 0
       0      .1       0   485.6    .045       0   500.6      .1       0
Bank Sta=485.6,500.6
XS Rating Curve= 0 ,0
Exp/Cntr=0.3,0.1

Type RM Length L Ch R = 1 ,22235.7 ,316.151,321.21,326.269
XS GIS Cut Line= 3
     1732235.743      351623.535      1731790.91      351519.501
     1731294.778      351317.678
#Sta/Elev= 30
       0  1102.8    77.8  1080.6   106.9 1069.25   126.4 1059.03   145.8 1053.12
   194.4 1027.92   204.1 1024.97   223.6 1010.39   233.3 1008.61   252.7  996.56
   262.4  994.47     311  993.79   330.5  990.81   359.6  990.81   388.8  987.53
   495.8  987.53   520.9  984.96     525   984.9   535.9  986.39   622.4  999.04
   680.8 1033.42   700.3 1048.15     749  1070.5   787.9 1078.68   836.6 1097.14
   885.3 1109.07   924.3 1123.65     934 1130.16   943.8 1131.97   992.4  1153.5
#Mann= 3 , 0 , 0
       0      .1       0   520.9    .045       0   535.9      .1       0
Bank Sta=520.9,535.9
XS Rating Curve= 0 ,0
Exp/Cntr=0.3,0.1

Type RM Length L Ch R = 1 ,21914.5 ,340.087,335.165,330.243
XS GIS Cut Line= 3
     1732274.648       351334.93     1731830.371       351221.75
      1731405.87      350958.131
#Sta/Elev= 30
       0 1118.28    19.5 1109.33    87.8 1090.39   136.6 1067.94   185.3 1050.91
   204.8 1035.86   224.4 1026.56   234.1 1018.12   253.6 1009.29   263.4 1002.33
   282.9  996.16   331.7  990.81   390.2  990.81   419.4  987.64   505.5  984.52
   507.5  984.32   520.5  985.97   605.4  997.11   664.2 1033.01   713.2 1049.96
   752.4 1059.96   781.8 1071.82   791.6 1072.07   811.2 1078.77   830.8  1080.6
   840.6 1083.53   850.4    1090   899.4 1095.34   928.8 1104.79   958.2 1108.27
#Mann= 3 , 0 , 0
       0      .1       0   505.5    .045       0   520.5      .1       0
Bank Sta=505.5,520.5
XS Rating Curve= 0 ,0
Exp/Cntr=0.3,0.1

Type RM Length L Ch R = 1 ,21579.4 ,469.383,487.842,506.301
XS GIS Cut Line= 3
     1732412.999      351112.653     1731868.038      350906.062
     1731493.158      350854.045
#Sta/Elev= 30
       0 1077.72    77.7 1059.23    87.4 1058.49   126.3 1045.05   155.4  1038.6
   174.8 1036.61   184.6  1033.5   213.7 1020.37   233.1 1005.51   252.5   995.2
   301.1  990.81     340  990.76   359.4  987.84   456.5  987.45   532.7  981.05
   534.2  980.97   547.7  982.62     641   994.1   660.4  995.11   670.1  997.37
   757.5 1000.88   776.9 1007.43   786.6 1009.05     806 1017.82   815.7  1020.1
   835.1 1029.45   864.2 1034.18   883.6 1034.06   912.8 1037.45   961.3 1049.48
#Mann= 3 , 0 , 0
       0      .1       0   532.7    .045       0   547.7      .1       0
Bank Sta=532.7,547.7
XS Rating Curve= 0 ,0
Exp/Cntr=0.3,0.1

Type RM Length L Ch R = 1 ,21091.5 ,310.139,311.559,312.98
XS GIS Cut Line= 3
     1732535.657      351016.278     1732202.728      350630.782
     1731993.624      350164.446
#Sta/Elev= 30
       0 1092.94    19.6  1088.6      98 1056.66   127.3 1047.93   244.9   991.9
   303.7  990.61   323.2  987.53     431  987.53   460.4  984.32     529  984.25
     552  981.48   558.5  980.97     567  982.05   597.8 1005.38   617.5 1013.14
   637.1 1025.94   656.8 1033.63   686.3 1053.34   705.9 1060.16   764.9 1088.01
   794.4    1098     814  1108.5   823.9 1109.16     873 1123.46   902.5 1138.27
   912.3 1139.34   941.8 1155.99   981.1 1173.33  1000.8 1179.44  1020.4 1189.65
#Mann= 3 , 0 , 0
       0      .1       0     552    .045       0     567      .1       0
Bank Sta=552,567
XS Rating Curve= 0 ,0
Exp/Cntr=0.3,0.1

Type RM Length L Ch R = 1 ,20780   ,791.689,838.795,843.682
XS GIS Cut Line= 3
     1732640.792      350893.621     1732412.999      350367.944
     1732202.728      349964.924
#Sta/Elev= 30
       0 1104.15    19.4 1098.58    48.6 1085.98   106.8 1069.45   126.2  1059.1
   155.4 1050.09   184.5 1037.12   213.6 1013.26   223.3 1010.93   242.8  999.68
   271.9  988.91     369  984.25     437  984.25   466.1  980.97   537.5     981
   543.8  981.05   552.5  983.71   592.3 1003.01   611.6  1010.1   640.6  1035.2
   679.3 1061.29     718 1075.76   737.3 1078.88   785.7 1090.73     805 1098.27
   824.4 1100.21   872.7 1113.68   911.4 1121.69   940.4 1131.21  1027.5 1133.62
#Mann= 3 , 0 , 0
       0      .1       0   537.5    .045       0   552.5      .1       0
Bank Sta=537.5,552.5
XS Rating Curve= 0 ,0
Exp/Cntr=0.3,0.1

Type RM Length L Ch R = 1 ,19941.2 ,556.583,533.671,512.661
XS GIS Cut Line= 3
      1733077.69      350699.719     1732934.862      350239.493
     1732535.657      349842.266
#Sta/Elev= 30
       0 1041.23    49.2 1036.52   108.2  1036.8   167.2 1024.13   186.9 1022.81
   206.5 1015.65   216.4 1015.25   245.9 1001.74   265.5 1000.19     295  990.64
     354   987.3   393.4  981.18   422.9  980.97   449.5  977.31   452.4  977.01
   464.5  977.15   491.6  980.48   540.1  981.28   549.8  983.78   608.1  984.36
   666.4  990.69   734.3  994.36   773.2 1000.25   947.9 1000.77   957.7 1002.31
   977.1 1013.16   986.8 1016.01   996.5 1015.99  1025.6 1026.52    1045 1028.66
#Mann= 3 , 0 , 0
       0      .1       0   449.5    .045       0   464.5      .1       0
Bank Sta=449.5,464.5
XS Rating Curve= 0 ,0
Exp/Cntr=0.3,0.1

Type RM Length L Ch R = 1 ,19407.5 ,295.298,301.028,302.983
XS GIS Cut Line= 3
     1733480.309      349989.568     1733171.793      349859.795
     1732608.196      349649.085
#Sta/Elev= 30
       0 1044.93    47.8 1054.09    76.5 1054.66    86.1 1053.02   105.2 1047.87
   143.4 1041.69   210.4 1019.66   229.5 1015.01   258.2  999.31     306  977.97
   334.7  977.64   383.2  973.08   384.8  973.27   399.8  974.36     422  974.71
   431.7  976.81   460.9  977.86   470.6  980.19   509.4  983.98   567.6  987.53
   577.3  990.49     587  990.81   645.3 1000.65   674.4 1000.74   693.8  1003.9
   790.8 1003.93   849.1 1000.65   887.9 1005.81     917 1021.79   936.4 1038.72
#Mann= 3 , 0 , 0
       0      .1       0   384.8    .045       0   399.8      .1       0
Bank Sta=384.8,399.8
XS Rating Curve= 0 ,0
Exp/Cntr=0.3,0.1

Type RM Length L Ch R = 1 ,19106.5 ,381.286,392.337,409.13
XS GIS Cut Line= 3
     1733458.272        349935.7     1733299.117      349617.389
     1732821.237      349466.025
#Sta/Elev= 30
       0 1041.47    28.9 1037.04    48.1 1037.27    86.6 1029.61     125  1017.9
   163.5  996.42   173.1  994.01   182.8  987.57   192.4  983.06     202  981.06
   250.1   980.8   278.9  977.83   346.3  977.69   375.5  971.85   385.4  971.13
   386.9  971.13   401.9  971.13   434.5  971.32   454.2  974.41   513.1  974.64
   532.8  977.69   552.5  977.69   621.3  995.17   660.6 1000.22   778.5 1000.94
   788.4 1004.06     808 1017.54   827.7 1036.94   837.5 1043.34   857.2 1053.34
#Mann= 3 , 0 , 0
       0      .1       0   386.9    .045       0   401.9      .1       0
Bank Sta=386.9,401.9
XS Rating Curve= 0 ,0
Exp/Cntr=0.3,0.1

Type RM Length L Ch R = 1 ,18714.1 ,409.359,421.41,425.241
XS GIS Cut Line= 3
     1733797.282      349903.595      1733482.63      349421.974
     1733299.315      348938.295
#Sta/Elev= 30
       0 1085.05    29.3 1077.14    68.3 1062.93   146.3 1047.33   175.5 1035.41
     195 1032.63   224.3 1018.01   243.8 1013.38     273  999.32   321.8  987.54
   458.3  978.11   516.8  977.69     546  971.47   567.8  970.48   582.8  969.59
   585.1  969.53   633.9  971.56   663.1  975.88   711.9  996.19   721.7  998.36
   770.5 1003.93   799.8 1004.11     829 1010.06   868.1 1024.47   907.1 1043.83
   936.4 1062.08   946.2 1062.97   985.2 1079.77  1024.2 1091.48  1092.5 1122.68
#Mann= 3 , 0 , 0
       0      .1       0   567.8    .045       0   582.8      .1       0
Bank Sta=567.8,582.8
XS Rating Curve= 0 ,0
Exp/Cntr=0.3,0.1

Type RM Length L Ch R = 1 ,18292.7 ,350.605,358.54,366.474
XS GIS Cut Line= 3
     1733972.508      349807.221     1733744.714       349316.59
     1733495.662      348815.161
#Sta/Elev= 30
       0 1111.13    39.3 1097.34      59  1087.8    68.8 1086.23     118 1067.52
   167.2 1053.82     236 1030.61   245.9 1029.53   285.2 1012.39   324.6 1000.97
   413.1     991   472.1  990.33   531.1  977.69   648.3  968.72   658.8  967.85
   663.3  969.31   678.4  972.28   698.1  979.93     757  997.17   776.7 1000.74
   796.3  1009.9     816 1014.67   845.4 1028.39   894.5  1043.1   933.8 1059.74
   943.6 1060.64   982.9  1076.8  1012.4 1093.19  1071.3 1116.67  1100.8 1133.12
#Mann= 3 , 0 , 0
       0      .1       0   648.3    .045       0   663.3      .1       0
Bank Sta=648.3,663.3
XS Rating Curve= 0 ,0
Exp/Cntr=0.3,0.1

Type RM Length L Ch R = 1 ,17934.2 ,435.12,420.05,407.048
XS GIS Cut Line= 3
     1734156.495      349772.176     1734042.598      349193.932
     1733988.488      348662.498
#Sta/Elev= 30
       0 1091.78   147.3 1057.55     167 1055.69   225.9 1038.37     275 1029.17
   343.8 1008.32   432.2  986.63   451.8   977.8     501  974.44   599.1  974.41
   618.5  971.13   664.6  968.68   676.8  967.85   679.6  967.87   715.6  972.26
   754.5  986.93   773.9 1000.22   793.3 1007.11   812.7 1019.41   832.2 1026.66
   861.3 1045.31   900.2 1061.23   948.7 1073.51   977.9 1084.54   997.3 1085.95
  1026.4 1096.45  1055.5 1111.34  1065.3 1112.91  1094.4 1127.78  1123.5 1136.16
#Mann= 3 , 0 , 0
       0      .1       0   664.6    .045       0   679.6      .1       0
Bank Sta=664.6,679.6
XS Rating Curve= 0 ,0
Exp/Cntr=0.3,0.1

Type RM Length L Ch R = 1 ,17514.1 ,404.734,400,405.093
XS GIS Cut Line= 3
     1734796.068      349421.725     1734427.844      349043.249
     1734091.381      348627.239
#Sta/Elev= 30
       0 1060.74    19.6  1059.2    97.8 1041.17   117.3 1039.94   205.4 1017.47
   234.7  1006.1     264  998.36   283.6  997.18   400.9  977.71   469.4  977.68
   520.5  965.26     528  964.57   535.5  964.57   644.8  980.56   722.6  984.94
   751.8  989.17   761.5  991.87     781 1002.69   800.4 1007.16   829.6 1022.67
   858.8 1030.76   878.3 1041.06   897.7 1044.67   926.9 1058.64   956.1 1066.99
   975.5 1076.48     995  1080.2  1024.2 1094.55  1043.6 1099.24  1063.1  1107.6
#Mann= 3 , 0 , 0
       0      .1       0   520.5    .045       0   535.5      .1       0
Bank Sta=520.5,535.5
XS Rating Curve= 0 ,0
Exp/Cntr=0.3,0.1

Type RM Length L Ch R = 1 ,17114.1 ,396.559,400,391.713
XS GIS Cut Line= 3
     1734983.049      349006.521     1734590.537         348710.
     1734388.356      348307.969
#Sta/Elev= 30
       0 1076.04    19.7 1069.58    39.4 1065.94    88.5 1047.14    98.4 1046.61
   137.7 1028.99   167.3  1020.6   216.4  998.07   265.6  986.58   295.2  970.17
   314.8  967.85   423.1  967.85   442.7  964.98   484.4  963.87   491.9   962.9
   499.4  964.69   560.4  987.05     580  990.67   599.5  996.58   628.9 1001.09
   697.4 1015.82   716.9 1021.82   736.5 1029.53   756.1 1034.59   775.6 1044.17
   844.1 1068.02   863.7 1077.12   883.2 1082.82   912.6 1096.64   941.9  1107.4
#Mann= 3 , 0 , 0
       0      .1       0   484.4    .045       0   499.4      .1       0
Bank Sta=484.4,499.4
XS Rating Curve= 0 ,0
Exp/Cntr=0.3,0.1

Type RM Length L Ch R = 1 ,16714.1 ,426.585,423.34,419.928
XS GIS Cut Line= 3
     1735217.863      348746.714     1734877.896      348443.143
      1734540.87       348137.67
#Sta/Elev= 30
       0 1063.45    48.5  1045.1    67.9 1040.55      97 1027.41   116.4  1022.9
   145.5 1008.62   184.3  995.27   203.6   986.3   232.7  982.35   252.1  971.18
   261.8  968.31   310.3  967.69   339.4  964.57   407.3  964.36   426.7  961.28
   448.3   961.4   463.3  963.14   475.1  965.41   542.9  991.68   571.9  997.88
   610.6 1010.22     630 1018.69   649.3 1022.08     659 1026.82   765.5 1060.64
   784.8 1069.86   804.2 1075.21   833.2 1086.87   891.3 1103.19   910.6 1111.77
#Mann= 3 , 0 , 0
       0      .1       0   448.3    .045       0   463.3      .1       0
Bank Sta=448.3,463.3
XS Rating Curve= 0 ,0
Exp/Cntr=0.3,0.1

Type RM Length L Ch R = 1 ,16290.8 ,180.218,178.467,176.856
XS GIS Cut Line= 3
     1735568.405      348414.637     1735161.239      348131.235
     1734738.484      347851.851
#Sta/Elev= 30
       0 1028.08    19.5 1028.79    48.6 1025.47    77.8 1016.46   136.2 1003.61
   233.5  987.36   262.6  976.51   272.4  974.81   311.3  973.68     321  971.13
   340.5  971.13   359.9  967.85   398.8  967.83     428  964.58   505.8   964.4
   534.4  961.37   535.1  961.29   549.4  962.66   642.3  974.87   681.2  984.69
   700.7  991.67   749.5 1001.53   768.9 1009.37   817.7 1023.14   846.9 1037.21
   866.4 1042.42   876.1 1048.82   895.6 1056.35   924.9 1071.65  1002.8 1095.08
#Mann= 3 , 0 , 0
       0      .1       0   534.4    .045       0   549.4      .1       0
Bank Sta=534.4,549.4
XS Rating Curve= 0 ,0
Exp/Cntr=0.3,0.1

Type RM Length L Ch R = 1 ,16112.3 ,176.246,179.175,182.616
XS GIS Cut Line= 3
     1735768.571      348554.358     1735348.029      348054.965
     1734874.645      347729.323
#Sta/Elev= 30
       0 1015.91    19.5 1017.35    48.7 1013.47    68.2  1015.3    87.7 1010.38
   116.9 1013.13   146.2 1007.81   165.7  1010.8   194.9 1006.42   243.6 1006.23
   263.1 1009.03   292.3 1003.83   360.5 1000.65     458  984.76   506.7  980.81
   555.4  971.16   604.2   970.7   750.3  961.28   793.3  961.28   808.3  961.28
   886.6  966.54   915.8  972.94   954.8  978.17  1003.5  990.38  1032.7  994.96
  1100.9 1018.26  1120.3 1027.03  1139.8 1031.99    1169 1046.02  1227.5 1065.81
#Mann= 3 , 0 , 0
       0      .1       0   793.3    .045       0   808.3      .1       0
Bank Sta=793.3,808.3
XS Rating Curve= 0 ,0
Exp/Cntr=0.3,0.1

Type RM Length L Ch R = 1 ,15933.2 ,426.708,434.102,440.165
XS GIS Cut Line= 3
     1735772.885      348242.443     1735419.529      347926.755
     1734899.361      347566.225
#Sta/Elev= 30
       0  976.09     9.7  974.41   125.7  974.41   135.4  976.82   174.1  978.92
   212.7  985.56   241.8  987.52   299.8  984.38   309.4  982.64   328.8  974.68
   348.1  971.13   415.8  971.13   425.5  968.84   464.2  967.59   483.6  964.57
     542  964.25   571.2  961.28   613.1  961.28   628.1  961.28   649.1  961.35
     688  967.85   717.3  967.85   775.7  976.84   804.9  977.81   814.6  980.16
   863.3  980.97   921.7  993.04  1028.8 1010.44  1087.3 1011.14  1106.7 1013.26
#Mann= 3 , 0 , 0
       0      .1       0   613.1    .045       0   628.1      .1       0
Bank Sta=613.1,628.1
XS Rating Curve= 0 ,0
Exp/Cntr=0.3,0.1

Type RM Length L Ch R = 1 ,15499.1 ,388.702,384.915,384.454
XS GIS Cut Line= 3
     1735851.807      347838.865     1735500.245      347562.638
     1735128.953      347160.853
#Sta/Elev= 30
       0   982.4    19.4   978.4    48.6  977.74    87.5  980.84   106.9  980.34
   126.4  975.88     175  968.01   213.8  967.42   233.3  964.57   388.8  964.57
   408.2  961.86   447.1  961.28   589.1  961.28   604.1  961.33   622.9  964.01
   652.3  966.11   671.8  976.44   681.6  979.85   710.9  983.98   720.6  984.25
   740.2  989.04   759.7  991.86     789  998.42   798.8  997.83   808.6  998.87
   837.9 1005.97   857.4 1004.92   886.7 1000.63     916 1000.66   994.2 1010.46
#Mann= 3 , 0 , 0
       0      .1       0   589.1    .045       0   604.1      .1       0
Bank Sta=589.1,604.1
XS Rating Curve= 0 ,0
Exp/Cntr=0.3,0.1

Type RM Length L Ch R = 1 ,15114.1 ,419.245,423.108,423.758
XS GIS Cut Line= 3
     1736224.158      347809.649     1735694.107      347293.837
     1735397.851      346934.547
#Sta/Elev= 30
       0 1059.78    19.5 1056.87     107 1031.94   126.5 1029.22     146 1023.95
   184.9 1016.91   214.1 1013.03   282.2  996.34   301.7  993.65   330.9   985.1
   369.8   981.2   389.3  975.42   437.9  964.69   457.4  961.75   486.6  964.05
   554.7  961.28   732.1  961.31   747.1  962.85     759  968.17   778.4  973.62
   807.5  977.44   865.7  977.89   923.9  984.25   943.3  984.25   982.1  990.34
  1040.4  994.49  1098.6 1001.36  1137.4  1010.5  1147.1  1010.5  1205.3 1025.33
#Mann= 3 , 0 , 0
       0      .1       0   732.1    .045       0   747.1      .1       0
Bank Sta=732.1,747.1
XS Rating Curve= 0 ,0
Exp/Cntr=0.3,0.1

Type RM Length L Ch R = 1 ,14691   ,333.258,327.321,321.247
XS GIS Cut Line= 3
     1736338.054      347555.571     1735946.872      347074.756
     1735674.232       346818.26
#Sta/Elev= 30
       0 1068.27    49.2 1055.34    78.7 1045.39    98.4 1041.81   118.1 1035.07
   137.7 1031.73   167.3 1021.68   236.1 1006.26   314.8  983.36   344.4  980.24
   354.2  977.28   373.9  967.55   393.6   962.2   482.1  960.99   501.8     958
   560.3   958.2   570.7  960.22   575.3  963.24   600.2  978.59   629.4  986.76
   658.2   988.5   696.6  993.48   725.4  994.19   744.6  997.37   773.4  997.37
   792.6 1000.09   821.4 1000.88   840.6 1003.93   869.4 1004.63   994.2 1021.98
#Mann= 3 , 0 , 0
       0      .1       0   560.3    .045       0   575.3      .1       0
Bank Sta=560.3,575.3
XS Rating Curve= 0 ,0
Exp/Cntr=0.3,0.1

Type RM Length L Ch R = 1 ,14363.7 ,439.165,449.571,466.641
XS GIS Cut Line= 3
      1736624.94      347208.744     1736219.511      346924.087
      1735887.68      346816.466
#Sta/Elev= 30
       0 1078.63    29.1 1067.93    48.6 1059.02      68 1052.88    87.4 1044.23
    97.1 1042.31   106.8 1038.12   126.3 1032.57   155.4  1025.1   194.3 1017.06
     204 1016.87   281.7  1002.7   310.8  994.65     340  982.06   349.7   979.7
   359.4  975.65   388.5  971.25   446.8     958   448.7     958   463.7  958.41
   534.1  978.68   553.5  982.83   572.9  984.28   621.4  993.59   660.1  994.44
   679.5  997.12   727.9  997.78     757 1000.65   824.8 1000.65   844.2 1003.66
#Mann= 3 , 0 , 0
       0      .1       0   448.7    .045       0   463.7      .1       0
Bank Sta=448.7,463.7
XS Rating Curve= 0 ,0
Exp/Cntr=0.3,0.1

Type RM Length L Ch R = 1 ,13914.1 ,406.348,402.608,392.204
XS GIS Cut Line= 3
     1736762.996      347061.686     1736535.068      346643.105
     1736440.735      346201.891
#Sta/Elev= 30
       0 1076.96    48.6  1060.8    68.1 1057.41    87.5 1051.04   155.6 1034.02
   175.1 1025.15     214 1017.29   233.4 1010.37   243.2 1009.51   272.4 1000.77
     321  980.92   330.7  980.33   350.2  974.64   369.6  973.45   469.1  957.44
   476.6   955.1   484.1  957.22   515.8  963.69   555.1  976.67   564.9  982.29
   584.5  987.21   604.1  994.73   623.7  999.03   682.6 1019.22     712 1023.38
   780.7 1023.89   819.9 1035.14   849.3 1045.58   898.4 1054.11   927.8 1065.26
#Mann= 3 , 0 , 0
       0      .1       0   469.1    .045       0   484.1      .1       0
Bank Sta=469.1,484.1
XS Rating Curve= 0 ,0
Exp/Cntr=0.3,0.1

Type RM Length L Ch R = 1 ,13511.5 ,364.644,373.324,382.005
XS GIS Cut Line= 3
     1737245.437      346878.169     1736938.285      346550.226
     1736638.926      346167.493
#Sta/Elev= 30
       0 1058.72    48.8  1060.7    68.4 1064.12    97.7 1064.27   166.1    1049
   185.6 1040.68   205.1 1036.91   263.7 1015.81   312.6  1008.6   361.4  998.27
   371.2   994.2   390.7  981.08   410.2  975.68   429.8  973.32   473.8  956.19
   488.2  954.72   488.8  954.72   565.9  958.86   643.7  980.16   663.1  983.81
   692.3  995.09   721.4 1003.56   740.9  1012.4   760.3 1015.84   789.5 1029.66
   847.8  1043.2   857.5 1041.97   867.2 1043.59   906.1  1053.1   935.2 1063.49
#Mann= 3 , 0 , 0
       0      .1       0   473.8    .045       0   488.8      .1       0
Bank Sta=473.8,488.8
XS Rating Curve= 0 ,0
Exp/Cntr=0.3,0.1

Type RM Length L Ch R = 1 ,13138.2 ,426.047,424.067,415.762
XS GIS Cut Line= 3
     1737328.007      346841.578     1737139.671      346197.646
     1736858.062      345939.355
#Sta/Elev= 30
       0 1014.09    48.6 1013.41    97.2 1009.23   116.7 1010.68   184.7 1005.37
   243.1 1003.84     282  999.32   301.4  994.15   320.9  991.83   340.3  985.26
   359.8  983.92   388.9  978.24   437.5   974.2     457  969.35   505.6  964.18
   515.3  961.28   599.9  953.28   614.9  952.28     632  951.44   661.2  953.44
   680.7  965.16   700.3  973.69   719.9  986.05   749.3  994.42   768.9 1003.14
   847.3 1021.83   866.9 1024.73   896.3 1033.28   994.2 1053.37    1053 1068.87
#Mann= 3 , 0 , 0
       0      .1       0   599.9    .045       0   614.9      .1       0
Bank Sta=599.9,614.9
XS Rating Curve= 0 ,0
Exp/Cntr=0.3,0.1

Type RM Length L Ch R = 1 ,12714.1 ,403.874,400,387.985
XS GIS Cut Line= 3
      1737608.44      346696.966     1737424.582      346085.299
     1737316.452      345646.804
#Sta/Elev= 30
       0 1036.55    78.6 1010.96   137.6 1001.45   186.7 1001.27   216.2   996.2
   245.7  987.21   265.3  985.54   294.8     991   383.2  990.36   412.7  986.75
   442.2  977.94   481.5   969.6     511  959.46   560.1   957.6   579.7  954.83
     619  954.72   631.2  952.19   638.7  951.44   646.2  951.44   697.6  958.44
   736.9  973.56   776.2  983.92   825.2  988.66   854.7  996.04   913.6  1007.3
   943.1 1010.67    1002 1021.54  1031.4 1024.41  1070.7 1034.31  1090.3 1044.68
#Mann= 3 , 0 , 0
       0      .1       0   631.2    .045       0   646.2      .1       0
Bank Sta=631.2,646.2
XS Rating Curve= 0 ,0
Exp/Cntr=0.3,0.1

Type RM Length L Ch R = 1 ,12314.1 ,400.9,400,395.688
XS GIS Cut Line= 3
     1737946.951      346335.466     1737711.552      345936.636
     1737498.407       345551.92
#Sta/Elev= 30
       0 1066.53     9.6 1065.65    48.2 1053.03    77.2 1037.65    96.5 1031.01
   135.1 1023.21     164 1012.23   183.3 1007.27     193 1006.46   212.3 1000.07
   279.8  987.33   299.1  982.07   318.4  980.39   385.9  961.54   405.2  960.78
   455.6  951.64   463.1  951.44   470.6  951.44   492.4  954.72   560.9  954.96
   570.6  956.77   609.7  968.39   707.5  991.58   746.6  1000.6   775.9 1004.82
   805.2 1013.18     815 1013.92   863.8 1031.23   893.2 1044.65   902.9 1046.48
#Mann= 3 , 0 , 0
       0      .1       0   455.6    .045       0   470.6      .1       0
Bank Sta=455.6,470.6
XS Rating Curve= 0 ,0
Exp/Cntr=0.3,0.1

Type RM Length L Ch R = 1 ,11914.1 ,376.887,387.363,399.08
XS GIS Cut Line= 3
     1738244.318      346079.951     1737908.182      345660.749
     1737614.125      345332.807
#Sta/Elev= 30
       0 1038.11    19.5 1033.88    39.1  1032.7   214.9  991.69   244.2  988.72
   263.8  984.77   332.2  980.97   341.9  978.71   361.5  967.49     381  963.41
   400.6  954.26   410.3  951.89   449.4  948.16   488.5  948.16     508  950.88
   529.8  951.44   544.8   951.5   556.9  953.26   576.5   963.5   615.6  977.09
   684.1  994.53   723.3 1006.77   742.9 1009.25   762.5 1017.51   791.8  1023.8
   840.8 1041.39   899.5 1066.56   938.6  1088.3   948.4 1091.04   977.8 1109.51
#Mann= 3 , 0 , 0
       0      .1       0   529.8    .045       0   544.8      .1       0
Bank Sta=529.8,544.8
XS Rating Curve= 0 ,0
Exp/Cntr=0.3,0.1

Type RM Length L Ch R = 1 ,11526.8 ,404.342,412.637,409.235
XS GIS Cut Line= 3
     1738353.149      346118.721     1738226.642      345440.712
     1737927.097      345148.341
#Sta/Elev= 30
       0 1043.48    19.4 1036.37    29.1 1035.32    48.6 1025.99    87.4 1014.15
   106.9 1013.32   145.7 1007.22   184.6 1000.25   213.7  992.35   281.7  982.36
   369.1  972.15   398.3  970.96   466.3  952.61   524.6  948.16   621.7  950.07
   632.5  948.48   647.5  948.29   689.7  953.63   709.2  962.58   728.6  977.17
   748.1  986.64   796.8  996.89   816.3  997.84   923.3 1020.56   933.1 1023.72
   962.3 1038.56   981.7 1043.13  1010.9 1055.84  1098.6 1088.29  1108.3 1093.69
#Mann= 3 , 0 , 0
       0      .1       0   632.5    .045       0   647.5      .1       0
Bank Sta=632.5,647.5
XS Rating Curve= 0 ,0
Exp/Cntr=0.3,0.1

Type RM Length L Ch R = 1 ,11114.1 ,397.347,400,407.521
XS GIS Cut Line= 3
     1738484.569      346197.573     1738521.296      345469.442
     1738374.852      345037.811
#Sta/Elev= 30
       0 1029.48    29.2 1025.77    48.6 1020.13   223.6  996.92   272.2  987.94
   349.9  980.65   388.8  974.88   476.3  971.13   534.6  964.95   612.4  963.86
   670.7  951.14   719.3  944.88   721.6  944.88   736.6  944.88   816.3  948.34
     826  950.99   855.1  970.77   874.5  986.75   884.2  990.45   893.9  991.37
     923 1004.76   942.4 1008.86   961.8 1017.18   981.2 1019.67  1010.3 1028.48
  1058.8 1033.72  1087.9 1040.62    1117 1042.95  1175.2 1052.06  1184.9 1051.75
#Mann= 3 , 0 , 0
       0      .1       0   721.6    .045       0   736.6      .1       0
Bank Sta=721.6,736.6
XS Rating Curve= 0 ,0
Exp/Cntr=0.3,0.1

Type RM Length L Ch R = 1 ,10714.1 ,422.897,400,400.171
XS GIS Cut Line= 3
     1738528.375      346302.708     1738830.329      345601.219
      1738959.22      345089.004
#Sta/Elev= 30
       0 1026.94    39.2 1015.78    88.1 1007.13   195.8  996.42   323.1  972.08
   489.6  963.37   518.9  966.16   646.2   954.8   675.6  954.47   744.1  944.88
   756.2  944.88   771.2  944.99   793.1  948.73   812.6  961.43     842  976.23
   910.4  996.09   939.8 1010.22   949.6 1011.72   969.1 1022.26   988.7 1027.73
    1018 1042.19  1037.6 1044.05  1125.6  1064.2    1155 1067.13  1194.1 1074.92
  1213.7 1083.52  1233.2 1086.75  1262.6 1099.07  1272.3  1099.2  1291.9 1107.12
#Mann= 3 , 0 , 0
       0      .1       0   756.2    .045       0   771.2      .1       0
Bank Sta=756.2,771.2
XS Rating Curve= 0 ,0
Exp/Cntr=0.3,0.1

Type RM Length L Ch R = 1 ,10314.1 ,392.156,400,396.434
XS GIS Cut Line= 3
     1739427.507      346059.855     1739153.492       345738.49
     1739048.535      345107.003
#Sta/Elev= 30
       0 1082.37    39.3  1069.2    58.9 1060.44    78.6 1057.89     108 1047.63
   137.5 1040.59   147.3 1035.33   196.4 1017.22   206.3 1011.75   225.9 1005.61
   265.2   998.3   284.8  996.95   333.9   983.7   363.4  957.21   373.2  952.63
   392.9  950.64   414.8  945.27   429.8  944.88   480.5  944.88   509.6  948.16
   577.5  948.16   645.4  960.48   674.5  962.48   703.6  967.25   810.3  999.71
     820 1000.96   887.9 1020.72  1023.7 1055.98  1052.8 1072.48  1062.5  1073.5
#Mann= 3 , 0 , 0
       0      .1       0   414.8    .045       0   429.8      .1       0
Bank Sta=414.8,429.8
XS Rating Curve= 0 ,0
Exp/Cntr=0.3,0.1

Type RM Length L Ch R = 1 ,9914.1  ,397.494,400,393.985
XS GIS Cut Line= 3
     1739574.036      345962.036     1739378.686      345441.833
     1739318.952      345008.698
#Sta/Elev= 30
       0 1060.68    29.2 1047.43      39 1047.07     117 1023.08     156  1014.2
   175.5 1011.55     195 1004.99   253.5  990.93     312  970.29   331.5  966.27
   360.7  956.47   428.9  951.45   548.2  946.49   555.7  944.95   563.2  946.01
   652.8  951.44   691.7  962.26   720.9  977.84   740.3  984.47   759.7  994.65
   779.1 1000.99   798.6 1011.82     818 1018.46   837.4 1028.26   856.9 1033.66
   876.3 1043.19   934.6 1062.89   963.8 1079.19   973.5  1080.7   992.9 1092.59
#Mann= 3 , 0 , 0
       0      .1       0   548.2    .045       0   563.2      .1       0
Bank Sta=548.2,563.2
XS Rating Curve= 0 ,0
Exp/Cntr=0.3,0.1
